HEC-RAS study HACKERSCK.prj: HACKERSCK

--- HACKERSCK.g01 (geometry) --- (continued)

Type RM Length L Ch R = 1 ,22403   ,122.1,125.4,127.1
XS GIS Cut Line= 2
2180931.65496456754187.2991613842180995.99370739754905.458642125
#Sta/Elev= 30
       0 1111.81      34 1105.35    62.1 1096.73    70.2 1094.76   102.3  1091.6
   130.4 1090.92   174.6 1091.61   343.2  1090.7   443.6 1090.88   496.1 1090.37
     520 1090.81     524 1090.68   529.3 1089.13     536 1088.25  540.72 1089.13
   544.1 1090.22   556.1 1090.87   560.1 1092.27   568.1 1097.53   573.5  1100.1
   576.2 1100.74   588.3  1100.5   596.3 1102.54   636.4    1122   648.5 1123.23
   668.5 1122.36   672.6 1124.68   680.6 1131.68   688.6 1135.84     721 1144.93
#Mann= 5 ,-1,0
       0     .05       0     410     .06       0   529.3    .045       0
  540.72     .06       0     700      .1       0
Bank Sta=529.3,540.72
XS Rating Curve= 0 ,0
Exp/Cntr=0.3,0.1

Type RM Length L Ch R = 1 ,22277   ,33.4,33.3,34.1
XS GIS Cut Line= 6
2180635.30873413754255.9404367462180673.20998989754396.706962678
 2180866.4289792754622.7972323212180871.23941047754655.668512659
2180856.80811666754740.6527984112180894.41149678754887.570250259
#Sta/Elev= 30
       0 1098.16    30.3 1097.93     109    1096   162.4 1094.09   198.9 1092.08
   247.4 1090.53   416.4 1090.06   515.1 1090.57   520.9 1090.41   526.8 1089.67
   531.6 1088.37   535.5 1088.42  543.13 1089.68   551.6 1090.91   571.9 1091.34
   588.3 1092.25   592.4 1093.21   596.6 1095.38   600.7 1098.15   621.4 1107.49
   625.5    1110   633.8 1115.94   645.5 1122.92   658.6 1131.56   662.7 1132.13
   675.1 1131.99   691.7 1130.77   695.8 1130.95   701.2 1133.98   714.8 1143.81
#Mann= 9 ,-1,0
       0     .05       0      40     .06       0     140     .05       0
  255.78     .06       0  404.41     .05       0   526.8    .045       0
  543.13     .05       0  615.32     .06       0  714.82      .1       0
Bank Sta=526.8,543.13
XS Rating Curve= 0 ,0
Exp/Cntr=0.3,0.1

Type RM Length L Ch R = 1 ,22244   ,205.9,198.2,185.4
XS GIS Cut Line= 6
2180598.68069251754272.2445856942180636.58194828754413.011111626
2180829.80093758754639.1013812682180834.61136885754671.972661607
2180820.18007505754756.9569473582180857.78345517754903.874399207
#Sta/Elev= 30
       0 1098.87   112.8 1095.15   145.8 1093.51   205.9 1091.85     231  1090.2
   351.7 1089.83   385.2 1089.41   401.6 1090.16   423.5  1089.9     470 1090.19
   494.4 1090.09     4971089.649   503.7 1088.14   514.1 1089.64   518.9 1090.19
     556 1091.13   567.5 1092.15   575.7 1094.09   586.8  1098.2   616.3 1111.01
   642.5 1124.82   654.1 1132.22   658.9  1133.6   666.5  1134.6   674.8 1134.35
   687.2 1133.19   688.4 1133.38   691.4 1134.24   699.6 1140.92   714.8 1147.74
#Mann= 10 ,-1,0
       0     .05       0      20     .06       0     130     .05       0
  315.78     .06       0  384.41     .05       0     497    .045       0
   514.1     .05       0  595.32     .07       0  665.32     .06       0
  695.32      .1       0
Bank Sta=497,514.1
XS Rating Curve= 0 ,0
Exp/Cntr=0.3,0.1

Type RM Length L Ch R = 1 ,22046   ,483.8,491.9,483
XS GIS Cut Line= 4
2180329.30059342754360.5477649342180573.93274382754534.402382441
2180712.41836593754790.8573369512180749.96134216754931.804232082
#Sta/Elev= 30
       0 1114.16    18.2 1108.86    52.6 1100.89    91.4 1096.78   131.1  1095.3
   194.4 1094.94   307.8 1091.98   342.2 1089.89     354 1088.16   362.4 1088.88
   371.5 1087.62     376 1088.61   397.4 1089.32   489.7 1089.61   494.2 1087.83
   498.5 1087.29  512.57 1089.62   562.4 1089.85     576 1092.09   610.5 1102.51
   634.7 1106.06   656.1 1112.89   668.3 1118.69     685 1130.82   689.2 1133.07
   697.5 1134.78   705.7 1138.61   714.2  1139.1   733.8 1138.36   737.4 1139.95
#Mann= 5 ,-1,0
       0      .1       0     150     .05       0   489.7    .045       0
  512.57     .05       0  590.12     .06       0
Bank Sta=489.7,512.57
XS Rating Curve= 0 ,0
Exp/Cntr=0.3,0.1

Type RM Length L Ch R = 1 ,21554   ,487.7,497.3,489.6
XS GIS Cut Line= 3
2180238.91963004 754417.019804352180411.29341718754524.452769358
2180622.15065447754958.995060656
#Sta/Elev= 30
       0 1122.23    39.2 1115.76    82.3 1106.17   105.2 1099.97   121.3 1097.86
   133.5 1095.54   166.5 1093.26   243.9 1091.51   249.2 1091.07  267.76 1087.65
   283.9 1085.81   291.81087.643   297.3 1088.81   300.1 1088.84   388.4 1088.03
   487.8 1088.92   510.7 1090.66   524.6 1093.38   532.9 1096.31   541.8 1100.49
   546.3 1101.56   568.5 1104.02   595.2  1110.4   608.4 1111.59   621.8 1112.06
   626.4 1112.84   657.4  1125.4   675.2 1131.72   683.3  1139.8   686.1 1140.66
#Mann= 5 ,-1,0
       0      .1       0     140     .05       0  267.76    .045       0
   291.8     .05       0  603.11     .06       0
Bank Sta=267.76,291.8
XS Rating Curve= 0 ,0
Exp/Cntr(USF)=0,0
Exp/Cntr=0.3,0.1

Type RM Length L Ch R = 1 ,21056   ,196,196.5,194.6
XS GIS Cut Line= 2
2180090.66471851754536.8689590932180347.03582236755081.236127903
#Sta/Elev= 30
       0 1129.25    22.4 1121.63    71.1 1099.53    79.5 1097.96   109.6 1095.13
   118.6 1092.04   127.6 1086.75   139.6 1084.92  148.18 1086.75   155.1 1087.97
   175.7 1087.22   323.1 1086.91   362.9 1085.98   393.8 1087.25   407.1 1088.87
   431.2 1094.29   440.2  1097.8   446.9 1103.53   452.2 1106.31   473.4 1107.64
   486.7 1112.05     500 1113.47   508.8 1117.94   518.4 1121.71   530.9 1129.08
   548.6 1137.21     553  1138.1   575.1 1139.24   592.8 1138.86   601.7 1137.64
#Mann= 6 ,-1,0
       0      .1       0   127.6    .045       0  148.18      .1       0
     280     .05       0     500     .06       0     600      .1       0
Bank Sta=127.6,148.18
XS Rating Curve= 0 ,0
Exp/Cntr=0.3,0.1

Type RM Length L Ch R = 1 ,20860   ,343.9,351.1,355.3
XS GIS Cut Line= 3
 2179917.8189199754609.1404477932180182.50363902755111.128708177
     2180208.509      755161.277
#Sta/Elev= 30
       0 1144.76    40.3 1129.06    72.4 1123.85    81.7 1119.05    99.5 1106.42
   122.1 1097.84   140.2 1094.99   166.6 1087.72   176.4 1086.91   194.5 1087.39
   200.1 1086.27   208.1 1084.58   217.1 1085.08  220.45 1086.25   226.1 1088.33
   239.7 1086.77   257.8 1086.06   343.7    1087   405.8 1090.52   447.7  1094.5
   456.8 1097.31   474.9 1101.16   502.2 1108.96   542.7 1123.94   555.4 1133.23
   558.4 1134.42   565.3  1135.1   583.3 1134.61   601.3 1144.06     624 1150.01
#Mann= 6 ,-1,0
       0      .1       0   200.1    .045       0  220.45      .1       0
     300     .05       0     420     .06       0     510     .07       0
Bank Sta=200.1,220.45
XS Rating Curve= 0 ,0
Exp/Cntr=0.3,0.1

Type RM Length L Ch R = 1 ,20509   ,345.6,348.8,340.5
XS GIS Cut Line= 3
     2179712.386        754458.4 2179778.1171549755138.717605483
2180025.57714731755448.587786828
#Sta/Elev= 30
       0 1259.71    26.9 1250.76    63.1 1225.18    79.1 1216.46    91.2 1214.09
   119.3 1202.65   131.4 1200.08   187.6 1167.06   200.2 1160.97   276.1 1135.03
   292.1 1127.44   308.2 1123.11   348.4 1102.72   376.5 1086.17   508.1 1086.33
   517.2  1084.2  528.47 1086.31   533.7 1087.76   569.4 1088.17   621.7 1086.44
   637.7 1088.07   665.6 1086.25   840.4 1087.56   898.3 1090.62   957.9 1108.63
  1000.9 1106.86  1011.2 1110.02  1026.5 1118.57  1042.5 1120.11    1080 1134.27
#Mann= 6 ,-1,0
       0      .1       0   508.1    .045       0  528.47      .1       0
  823.49     .06       0  863.49      .1       0  973.49     .07       0
Bank Sta=508.1,528.47
XS Rating Curve= 0 ,0
Exp/Cntr=0.3,0.1

Type RM Length L Ch R = 1 ,20160   ,99.8,101.5,103.2
XS GIS Cut Line= 3
2179467.87861366754675.2780532562179565.18853778755177.904443295
2179255.85065728755389.448939601
#Sta/Elev= 30
       0 1145.75    22.3 1141.68    75.3 1126.91    95.6 1120.05   107.9 1114.59
   124.8 1109.82   152.7 1097.14   173.1 1090.56   185.3 1084.37   189.4 1083.51
  202.26 1084.37     212 1086.56   474.6 1084.75   576.2 1086.02   595.6 1083.75
     615 1087.09   631.1 1086.43   653.7 1091.77   702.1 1093.59   716.7 1095.97
   737.4 1095.47   765.2 1103.11   788.4 1114.53   802.8  1116.7   811.5  1119.4
   818.5 1123.49     833 1134.47   862.1 1150.73   871.9 1154.57   886.7 1156.89
#Mann= 8 ,-1,0
       0      .1       0   185.3    .045       0  202.26      .1       0
     420     .06       0     510      .1       0  521.96     .07       0
  641.96     .06       0  691.96      .1       0
#XS Ineff= 2 , 0
                          576.49         1095.71
Permanent Ineff=
       F       F
Bank Sta=185.3,202.26
XS Rating Curve= 0 ,0
Exp/Cntr=0.3,0.1

Type RM Length L Ch R = 1 ,20058   ,795.1,820.2,821
XS GIS Cut Line= 3
2179395.63056271754741.9496429942179413.88468127 755010.05700934
2179187.24346079755220.182822315
#Sta/Elev= 30
       0 1120.51    55.4 1108.82   107.5 1092.61   119.5    1088   123.5 1086.79
   131.2 1085.81   134.9 1084.21   139.6 1083.34   147.6 1083.21  151.59  1084.2
  151.59 1084.21   157.4 1086.24   163.6 1086.61   219.7 1085.49   247.8 1085.66
   320.2 1084.82   455.7  1085.1   464.6  1082.7   467.4 1082.72   475.9 1084.75
   484.4 1085.55   487.3 1086.87   494.7 1092.08   498.6 1093.52   521.2 1093.19
   524.1 1094.51   526.3 1096.22   532.5 1102.73   535.4 1104.07   577.8 1112.63
#Mann= 5 ,-1,0
       0      .1       0   134.9    .045       0  151.59      .1       0
  338.73     .06       0  518.73      .1       0
#XS Ineff= 2 , 0
                          455.07         1095.67
Permanent Ineff=
       F       F
Bank Sta=134.9,151.59
XS Rating Curve= 0 ,0
Exp/Cntr(USF)=0,0
Exp/Cntr=0.3,0.1

Type RM Length L Ch R = 1 ,19238   ,324.1,316.6,306.4
XS GIS Cut Line= 3
2179205.23935494754752.2254096662179159.85445797 754921.24502596
2178937.62496247 755048.00973818
#Sta/Elev= 30
       0 1105.34     9.3  1103.7    25.8 1099.59    42.4 1093.63    50.7 1091.22
    75.5 1087.98     129 1084.69   166.7 1085.31   206.9 1084.37   229.9  1084.9
   239.1 1084.56   243.7 1082.81   248.3 1081.82   253.9 1081.94  259.05 1082.81
   262.7 1084.35   266.7 1085.18   297.9 1084.42   326.6 1084.24     336 1084.59
   341.9 1086.11   352.5 1091.95   358.8 1093.41   368.6    1094   394.6 1093.12
   400.5 1094.27     409 1097.06   418.7 1097.21   423.3 1097.86   430.8 1096.95
#Mann= 6 ,-1,0
       0      .1       0     140     .07       0   243.7    .045       0
  259.05     .07       0  285.01     .06       0  395.01      .1       0
Bank Sta=243.7,259.05
XS Rating Curve= 0 ,0
Exp/Cntr(USF)=0,0
Exp/Cntr=0.3,0.1

Type RM Length L Ch R = 1 ,18922   ,245.2,246.5,246.7
XS GIS Cut Line= 4
2178999.50286847754569.6166917482178981.24874992754632.365224296
2178886.55550989755007.7155371742178787.87622391755103.972208652
#Sta/Elev= 30
       0 1123.81    31.4 1115.71    53.7  1109.1    82.7 1104.61   106.4  1101.6
   115.7 1098.89   136.3  1090.4   156.9 1086.17   161.1 1084.67   164.31082.844
   169.3 1081.62  180.39 1082.84   189.9 1084.15   231.2  1083.5   248.1 1084.27
   264.2 1083.33   327.2  1083.3   396.2 1084.31   400.3 1084.83   404.5 1086.59
   412.7 1091.69   416.8 1092.52   455.2 1092.19   460.3  1093.7   466.5 1097.39
   471.7 1099.65     475 1100.44   517.6 1105.98   534.8 1111.58   590.3 1123.86
#Mann= 5 ,-1,0
       0      .1       0   164.3    .045       0  180.39      .1       0
  325.35     .06       0  425.35      .1       0
Bank Sta=164.3,180.39
XS Rating Curve= 0 ,0
Exp/Cntr=0.3,0.1

Type RM Length L Ch R = 1 ,18675   ,252.4,253.6,251.2
XS GIS Cut Line= 4
2178785.16205057754508.6164323812178754.66626375754585.317956803
2178636.37957549754927.2404150692178593.94109831755051.256540992
#Sta/Elev= 30
       0  1126.3    24.3    1118      48 1110.74   106.4 1095.88   137.4 1084.37
   141.7 1083.49   145.9 1083.22   158.6 1083.59     1651081.809     167 1081.09
   169.3 1080.99   179.7 1081.81     184 1082.24   192.4 1083.87   213.6 1082.75
   217.8 1082.92   226.3 1084.16   247.9 1082.95   326.5 1083.33   408.3 1086.25
   430.3 1090.25     446 1090.35   454.9 1089.34   458.6 1089.55   471.8  1092.9
   480.2 1096.33   492.9 1099.27   526.7 1111.23   564.8 1121.07   575.4 1124.73
#Mann= 6 ,-1,0
       0      .1       0     165    .045       0   179.7      .1       0
  292.54     .06       0  402.54     .07       0  504.35      .1       0
Bank Sta=165,179.7
XS Rating Curve= 0 ,0
Exp/Cntr=0.3,0.1

Type RM Length L Ch R = 1 ,18421   ,225.6,227.9,226.5
XS GIS Cut Line= 2
2178541.86950265754443.069967885 2178409.7451784754966.864294065
#Sta/Elev= 30
       0 1119.33    68.2  1109.8    88.8 1103.97   105.3 1100.59   117.7 1096.85
   134.2  1090.2   142.4 1086.28   150.7 1083.34   158.9 1082.59   177.7 1083.33
     181 1082.95  186.21 1081.37   196.1 1080.63   204.41081.356   208.4 1082.38
     214 1082.89   240.3 1082.24   266.7 1083.36   336.3 1084.97   402.3 1085.56
   406.5 1086.06   418.2 1090.14   421.5  1090.7   444.6 1091.16   447.9  1092.1
   467.6 1101.43   472.5 1102.71   505.5 1106.41   530.2 1107.37   540.2 1109.84
#Mann= 6 ,-1,0
       0      .1       0  186.21    .045       0   204.4      .1       0
     250     .05       0     360     .06       0     460     .05       0
Bank Sta=186.21,204.4
XS Rating Curve= 0 ,0
Exp/Cntr=0.3,0.1

Type RM Length L Ch R = 1 ,18194   ,168.9,168.8,167.9
XS GIS Cut Line= 4
2178339.97875558754389.1582663732178316.97856619754466.728002309
  2178241.293568 754726.219424692178132.34043873754855.965135881
#Sta/Elev= 30
       0 1120.19    16.7 1119.36    33.4 1117.41    44.9 1114.67    66.8  1108.2
    87.6 1102.82   100.1    1101   116.8 1095.51   125.1 1092.02   137.6 1085.97
   151.3 1081.25   154.3 1080.25   157.7 1080.14   162.6 1080.29  167.96 1081.25
     171 1082.28   175.1 1082.87   204.3 1082.25   225.1 1082.62     246 1084.13
   295.1 1086.27   376.8 1088.09   412.5 1090.22   428.2 1091.57   442.1 1091.34
     462 1093.81   480.4 1098.09     496  1100.9   511.8 1102.38   520.6  1103.7
#Mann= 6 ,-1,0
       0     .05       0   151.3    .045       0  167.96     .05       0
  210.91     .07       0  310.91     .06       0  431.21     .05       0
#XS Ineff= 2 , 0
                          316.15         1090.64
Permanent Ineff=
       F       F
Bank Sta=151.3,167.96
XS Rating Curve= 0 ,0
Exp/Cntr=0.3,0.1

Type RM Length L Ch R = 1 ,18025   ,229.6,236.4,241
XS GIS Cut Line= 3
2178185.08214518754323.5357101872178164.60681871 754391.24284164
2178060.84005073754817.423705468
#Sta/Elev= 30
       0 1120.17    18.4 1117.32      56 1106.85    93.3 1097.98   105.7 1093.55
   113.9 1092.49   126.2 1088.56   134.5 1086.51   150.9 1083.66   167.4 1082.76
   171.5 1081.74     174 1080.57   175.6 1079.81   183.9 1080.09  185.75 1080.57
   192.1  1082.6   196.2 1082.94   220.9 1081.96   245.6  1082.2     268 1083.55
   278.6  1084.8   336.2 1086.16   381.5  1088.4   402.1 1090.22   410.4 1090.11
   414.4 1090.92     435 1099.29   451.5 1103.84   472.1 1108.73   509.4 1116.26
#Mann= 6 ,-1,0
       0     .05       0  170.74     .06       0     174    .045       0
  185.75     .06       0  380.74     .05       0  400.74      .1       0
Bank Sta=174,185.75
XS Rating Curve= 0 ,0
Exp/Cntr=0.3,0.1

Type RM Length L Ch R = 1 ,17788   ,151,152.7,153.5
XS GIS Cut Line= 4
2178078.61684381754273.2618239442178062.89765188754290.478081776
2177850.31429431754555.4587457892177761.77673322 754634.91278846
#Sta/Elev= 30
       0 1111.31    15.5 1109.22    26.8 1106.76    84.1 1090.33    93.4 1088.47
   142.7 1083.46   169.4 1082.41   206.3 1082.91   226.8 1081.82     245 1082.45
   247.3 1082.22   251.5 1080.55   257.5  1079.5  266.61 1080.55   271.9 1081.85
   286.1 1082.25   311.7 1087.64   321.7 1087.78   334.5    1087   337.3 1087.88
   344.7 1091.45     363 1098.73   377.1 1102.82   398.1  1111.5   411.1 1115.83
   419.6 1120.96     425 1123.15   459.2 1143.57   470.6 1148.87     482 1152.94
#Mann= 5 ,-1,0
       0     .05       0  153.31     .06       0   251.5    .045       0
  266.61     .06       0  303.31      .1       0
Bank Sta=251.5,266.61
XS Rating Curve= 0 ,0
Exp/Cntr=0.3,0.1

Type RM Length L Ch R = 1 ,17636   ,40.6,41.2,41
XS GIS Cut Line= 3
2178032.93897146754137.9426034692177813.60813783754365.589593747
2177643.77130494754535.983799841
#Sta/Elev= 30
       0 1121.67    15.6 1117.84    48.1 1114.83    64.5 1110.08   155.6 1090.08
   193.3 1083.17   209.3 1082.02   232.2 1082.19   243.3 1081.59     260 1082.28
   312.4 1082.55   319.7 1081.88   323.8 1080.68   332.5 1079.81   340.8 1080.56
  344.44 1081.84     348 1082.88   363.5 1084.56   384.7 1088.21   407.3 1087.22
   425.8 1096.15     430 1097.68   437.1 1098.92   449.8 1099.13     468 1104.58
   473.7 1106.92   499.5 1120.95   522.1  1134.7   544.8 1147.21   556.7 1150.85
#Mann= 5 ,-1,0
       0     .05       0   319.7    .045       0  344.44     .05       0
  346.12     .06       0  356.12      .1       0
Bank Sta=319.7,344.44
XS Rating Curve= 0 ,0
Exp/Cntr=0.3,0.1

Type RM Length L Ch R = 1 ,17594   ,220.2,230.5,229.6
XS GIS Cut Line= 3
2177992.06622484754122.3698031292177772.73539121754350.016793407
2177602.89855832754520.410999501
#Sta/Elev= 30
       0 1120.07     7.6 1118.19    47.2 1114.67    57.5 1112.05    98.3 1099.13
     132 1092.49   155.5 1086.13   168.8 1083.51   190.1 1081.81   276.6  1082.3
   291.71081.224   311.2 1079.57  330.91 1081.24   343.2 1082.05   354.5 1085.98
   367.9 1088.33   377.1 1088.62     394 1087.24   397.9 1087.55   407.6 1090.35
   418.9 1095.95   423.4 1097.44   435.9 1097.83   441.6 1098.77   467.4 1110.42
   484.4 1120.28   512.6 1134.07   525.2 1141.71   540.8  1149.8   556.7 1154.72
#Mann= 5 ,-1,0
       0     .05       0     290     .06       0   291.7    .045       0
  330.91     .06       0  376.12      .1       0
Bank Sta=291.7,330.91
XS Rating Curve= 0 ,0
Exp/Cntr=0.3,0.1

Type RM Length L Ch R = 1 ,17364   ,281.9,282,280.1
XS GIS Cut Line= 4
2177812.48486208754014.7549191922177769.05146873754072.974148573
2177560.20153476754360.3738364722177501.23185828754438.732175684
#Sta/Elev= 30
       0 1127.92    16.2 1118.32    30.5 1112.09    40.7 1109.35    62.9  1105.3
    76.3 1102.02    92.7 1096.38   127.3 1082.53     145 1081.43  149.95 1080.48
   156.9  1079.7   163.31080.475   171.8 1082.04   300.3 1081.52     330 1082.31
     335    1083   344.8 1088.04   351.2 1089.51   362.6 1089.85   380.3 1088.41
   384.4 1088.56   394.3  1092.1   404.2 1094.57   445.6 1110.61     459  1114.1
     464 1116.86   474.5 1125.61     504 1145.12   511.3 1148.61     526 1152.66
#Mann= 5 ,-1,0
       0     .05       0  149.95    .045       0   163.3     .05       0
  222.64     .06       0  372.64      .1       0
Bank Sta=149.95,163.3
XS Rating Curve= 0 ,0
Exp/Cntr=0.3,0.1

Type RM Length L Ch R = 1 ,17082   ,216.6,220.3,221.6
XS GIS Cut Line= 4
2177636.96650414753888.8090287632177583.36784852753976.599930211
2177440.13006194754229.807372282 2177377.5791102754350.127350883
#Sta/Elev= 30
       0 1120.33    29.9 1111.51    47.3 1109.18    61.4 1106.05    73.6 1104.91
      94 1100.58   117.4 1093.97   144.9 1085.23   163.3 1082.35   263.7 1080.82
   305.7 1081.83   317.91080.305   324.1 1079.63   331.6 1080.31   347.1 1081.94
   356.3 1083.69   370.1 1090.75   378.6 1092.95   393.1 1093.71   411.1 1092.69
   415.6 1092.99   424.6 1097.44   463.1 1109.63   470.4 1113.57   479.3 1120.03
   491.2 1132.79   500.1  1143.5     503 1145.99     506 1147.61   529.4 1156.33
#Mann= 6 ,-1,0
       0      .1       0      20     .05       0  242.86     .06       0
   317.9    .045       0   331.6     .06       0  352.86     .05       0
Bank Sta=317.9,331.6
XS Rating Curve= 0 ,0
Exp/Cntr=0.3,0.1

Type RM Length L Ch R = 1 ,16862   ,313,314.5,304.7
XS GIS Cut Line= 4
2177438.53232983753662.1971807532177370.23536793753961.206491273
2177263.87872632 754080.520731082177227.86451114754200.566437881
#Sta/Elev= 30
       0 1134.66    35.9  1124.2    76.9  1110.6    93.3 1106.54   111.3 1099.81
   114.7 1099.04   142.6 1096.22   154.9 1094.11   175.4 1088.45   191.5 1081.84
   195.9 1080.73   201.5  1080.3   249.2 1080.29   265.7 1081.29     312 1081.86
     328 1081.06     394 1081.17  400.42 1080.64   407.3 1079.69   413.8  1079.8
   418.6 1080.64   424.6 1081.72   467.2 1080.48   496.5  1081.4   513.2 1084.08
   554.9 1098.29   563.2 1099.71   567.5 1099.83   588.3 1097.85   591.9    1099
#Mann= 6 ,-1,0
       0      .1       0      40     .05       0  400.42    .045       0
   418.6     .05       0  486.55     .06       0  586.55     .05       0
Bank Sta=400.42,418.6
XS Rating Curve= 0 ,0
Exp/Cntr(USF)=0,0
Exp/Cntr=0.3,0.1

Type RM Length L Ch R = 1 ,16547   ,276.2,278.4,278.2
XS GIS Cut Line= 3
2177318.87386073753613.2900757322177150.20202143753928.028250106
2177075.42996895754241.027539538
#Sta/Elev= 30
       0 1112.94    40.7 1106.46    72.5 1099.25   131.5 1092.24   143.7 1089.97
   154.2 1088.89   176.9 1083.88   213.2 1083.91   267.6 1080.47   341.7 1081.17
   436.1 1080.49   489.9 1081.43   496.4 1080.26   502.2 1078.85   514.5 1078.68
   518.7 1078.96  521.21 1080.27   539.2 1089.13   551.6 1092.49   572.1 1101.43
   576.2 1102.31   588.8 1102.91   609.1 1103.02   613.2  1105.4   625.6 1115.66
   633.8 1123.86   637.9 1126.36   646.1 1129.95   654.4 1132.34   678.9 1141.56
#Mann= 5 ,-1,0
       0     .05       0   496.4    .045       0  521.21     .05       0
  537.09     .06       0  637.09     .05       0
Bank Sta=496.4,521.21
XS Rating Curve= 0 ,0
Exp/Cntr=0.3,0.1

Type RM Length L Ch R = 1 ,16269   ,511.5,517.6,506.7
XS GIS Cut Line= 4
2176986.31835917753237.0882826832176933.07718004753368.923583392
2176920.40070882753791.0500750852176903.92129623 754139.65303369
#Sta/Elev= 30
       0 1107.85      26 1103.92    64.8  1093.5    90.7 1090.02   127.7 1087.31
   267.6  1082.2   294.5 1081.53   318.5 1082.02   334.5 1080.89   374.5 1080.69
   394.5 1079.79   426.6 1080.46   438.6 1079.47   466.6 1080.56   502.6 1079.16
   526.6 1080.41   555.1 1080.04   654.7    1081   666.7 1080.93   673.8 1079.93
   682.8 1079.05  687.51 1079.93   706.8 1080.81   759.8  1080.3   786.9 1081.11
   794.9 1082.73   826.9 1096.46   850.9 1105.55     871 1106.34   913.5 1105.92
#Mann= 5 ,-1,0
       0     .05       0   673.8    .045       0  687.51     .05       0
   774.5     .06       0   874.5     .05       0
Bank Sta=673.8,687.51
XS Rating Curve= 0 ,0
Exp/Cntr(USF)=0,0
Exp/Cntr=0.3,0.1

Type RM Length L Ch R = 1 ,15751   ,39.8,39.9,40.3
XS GIS Cut Line= 6
2176886.73511879753220.4881704212176841.47880631753547.289382862
2176861.21750627753596.5358611752176853.07099867  753650.8459118
2176809.71609145753686.4664429882176719.33120913754095.995143417
#Sta/Elev= 30
       0 1090.65    61.3 1089.76   102.2 1087.71   178.4 1085.84   267.2 1082.27
   307.6 1082.75   323.8 1081.62   336.1 1081.52   351.9 1082.61   364.9 1080.95
  399.29 1079.98   409.4 1078.86   413.4 1078.99   417.6 1079.97   460.3 1080.69
     484 1080.18   624.1 1080.58   642.5 1080.12   687.6 1080.71   708.1 1081.76
     745    1082   781.7 1084.03   837.6 1089.39   880.1 1092.04   888.3 1093.37
   896.5 1095.86   900.6 1097.81   904.7 1100.42   908.8 1102.08   915.7 1103.07
#Mann= 5 ,-1,0
       0     .05       0  399.29    .045       0   417.6     .05       0
  716.36     .07       0  915.75     .05       0
Bank Sta=399.29,417.6
XS Rating Curve= 0 ,0
Exp/Cntr=0.3,0.1

Type RM Length L Ch R = 1 ,15711   ,281.1,283.7,278.1
XS GIS Cut Line= 6
  2176840.231493753224.4895373762176799.04843432753540.428739692
2176818.78713428753559.8046901622176814.71388048753641.269766099
2176771.35897325753676.8902972872176680.97409094754086.418997716
#Sta/Elev= 30
       0 1090.87    81.4 1088.17   155.2 1085.29   202.4 1084.25     279 1083.35
   307.6 1082.43   318.6 1081.75   325.8 1082.36   347.7 1081.27   363.8 1082.22
   384.1 1080.82  388.59 1079.89   392.1 1079.04   396.2 1078.75   404.3 1079.05
   410.41079.901   438.4 1081.01   484.7 1080.38   498.6  1080.6   514.6  1080.2
   569.1 1080.16   666.2 1081.43     710 1082.75   752.2 1086.24   800.6 1087.09
   809.5 1088.62   825.9 1089.19     871 1092.43   883.3 1094.75     905 1101.53
#Mann= 4 ,-1,0
       0     .05       0  388.59    .045       0   410.4     .05       0
  715.63     .07       0
Bank Sta=388.59,410.4
XS Rating Curve= 0 ,0
Exp/Cntr=0.3,0.1

Type RM Length L Ch R = 1 ,15428   ,260.5,277.1,287.2
XS GIS Cut Line= 3
2176609.60531722753159.064792424 2176578.0543643753369.610787243
2176505.64636068754096.074000034
#Sta/Elev= 30
       0 1091.78    54.7 1090.78   143.7 1087.08   189.5 1086.56   445.6  1080.8
   469.7 1079.92   473.8 1078.97   473.8 1078.95   481.8 1077.93   485.8    1078
   489.8 1078.92   493.9 1079.98   517.6 1080.14   538.1 1079.29   550.1 1080.25
   566.2 1079.45   582.3 1080.56   630.5 1081.06   666.7 1082.16   707.7 1084.09
   743.1 1086.96   755.2 1086.95   763.2 1085.73   787.3 1089.01   831.5 1092.62
   859.7 1094.01   891.8 1097.72   905.1 1101.47   919.7 1103.39     943 1103.29
#Mann= 6 ,-1,0
       0     .05       0   473.8    .045       0   489.8     .05       0
   752.9     .07       0   872.9     .06       0   942.9     .05       0
Bank Sta=473.8,489.8
XS Rating Curve= 0 ,0
Exp/Cntr=0.3,0.1

Type RM Length L Ch R = 1 ,15150   ,547.1,538.6,515.7
XS GIS Cut Line= 6
2176512.33586264753142.5857948552176503.20880336753208.756974634
 2176491.1661557753286.4637432252176454.15085973 753462.03286965
 2176119.7455489753642.6725845632176033.54554459753996.346131657
#Sta/Elev= 30
       0 1089.01      43 1087.13    95.6 1087.06   152.3 1084.98   248.2 1082.84
     292 1080.07   449.3  1080.1   455.6 1078.26   458.9 1077.65   466.1 1077.52
   473.81078.273   477.1 1079.45   481.7 1080.18     509 1079.88   523.5 1080.34
   558.9 1079.72   579.5 1078.34   595.3 1078.35   622.6 1079.44   682.9 1079.86
   740.5 1079.75   789.9 1078.34   855.2 1078.59   888.9  1080.6     934 1081.51
   950.4 1082.61   994.7 1087.36  1044.3 1094.68  1053.4 1096.73    1069  1098.1
#Mann= 7 ,-1,0
       0     .05       0  374.86     .07       0   455.6    .045       0
   473.8     .07       0  764.94     .05       0  974.94     .06       0
 1068.96     .05       0
Bank Sta=455.6,473.8
XS Rating Curve= 0 ,0
Exp/Cntr=0.3,0.1

Type RM Length L Ch R = 1 ,14612   ,285.1,281.3,278.4
XS GIS Cut Line= 4
2176076.91263656753068.1243624672176079.89639214753156.410104027
2176055.93786153 753565.986889212175959.49738991753976.360431473
#Sta/Elev= 30
       0 1117.46    80.6 1100.36   109.1 1093.62   121.2 1092.55   129.2 1090.41
   137.2  1088.8   145.2 1085.56  158.65 1078.73   161.2 1077.82   165.2 1077.31
   177.3 1077.38   185.3 1078.72   228.9 1079.72   273.4 1078.26   317.5 1078.34
   345.5 1078.85   368.9 1078.47   534.3 1078.37   567.5  1079.9   594.5 1080.03
   674.5 1079.45     769 1080.42   789.5 1081.23   814.2 1082.99   843.8 1086.22
   879.9 1091.18   896.4 1094.42   912.8 1095.52     917 1095.47   920.2 1094.99
#Mann= 7 ,-1,0
       0      .1       0  158.65    .045       0   185.3      .1       0
  248.34     .05       0  538.61     .07       0  638.61     .05       0
  738.61     .06       0
Bank Sta=158.65,185.3
XS Rating Curve= 0 ,0
Exp/Cntr=0.3,0.1

Type RM Length L Ch R = 1 ,14331   ,265.6,268.6,267.1
XS GIS Cut Line= 4
2175766.50481717753058.8674037912175777.95936704753110.011611028
2175879.48451211753749.3684778992175835.06208796753939.344961616
#Sta/Elev= 30
       0 1134.88    22.9 1129.27    59.7 1118.42    71.8 1113.28      92 1107.97
   112.3 1104.67   116.4 1102.95   128.5 1096.36   140.7 1091.94   152.8 1082.01
   156.9 1079.64   160.9 1078.62   177.1 1077.31  183.94 1078.61   189.3 1079.04
   213.6 1078.38   294.6 1080.06   403.9  1080.5   464.7 1078.19   535.9 1078.11
   602.2 1079.44   781.7 1080.24   810.5 1081.47   839.3 1084.71   843.4 1085.43
   855.5 1090.77   859.8 1091.55   876.2 1091.75   888.5 1090.35   894.9 1092.16
#Mann= 6 ,-1,0
       0      .1       0   160.9    .045       0  183.94      .1       0
  252.41     .05       0  759.78     .06       0  859.78     .05       0
Bank Sta=160.9,183.94
XS Rating Curve= 0 ,0
Exp/Cntr=0.3,0.1

Type RM Length L Ch R = 1 ,14062   ,287.1,302.9,297.4
XS GIS Cut Line= 3
2175530.38957356753116.456874357 2175610.6738913753571.401341546
2175524.48446045753805.669808147
#Sta/Elev= 30
       0 1124.66     4.8 1124.02      17    1124    29.2 1120.73    43.6 1119.79
    60.9    1116    73.8 1116.39    77.9 1115.81      82 1114.73      86 1112.76
    94.2 1106.96    98.2 1105.06   134.8 1094.65   175.4 1081.23   185.1 1079.39
   209.3 1078.25   224.1 1076.88   236.9 1078.24   260.7  1077.8   276.9 1078.35
   426.8 1078.58   506.5 1079.95   570.4 1084.36   658.5 1087.09   664.2 1087.96
   672.7 1090.92     677 1091.55   689.6 1092.22   702.5 1091.95   711.6 1095.28
#Mann= 7 ,-1,0
       0      .1       0     200     .05       0   209.3    .045       0
   236.9     .05       0  501.97     .07       0  601.97     .06       0
  711.59     .05       0
Bank Sta=209.3,236.9
XS Rating Curve= 0 ,0
Exp/Cntr=0.3,0.1

Type RM Length L Ch R = 1 ,13759   ,168.5,179,189.4
XS GIS Cut Line= 5
2175333.70848856753154.5600932562175295.81978373753225.716929166
2175311.52973451753405.9193058222175322.61911154753525.130108841
2175331.46052767 753679.77812801
#Sta/Elev= 30
       0 1104.34    21.1  1099.3    30.2 1096.63    62.8 1085.43    65.2  1084.9
    68.1 1084.49      80 1084.38   108.2  1080.3   123.6  1078.9   148.3 1078.13
   184.5 1078.36   189.6 1077.47   192.5 1076.91   200.5 1076.44   204.5 1076.54
   209.7 1077.46   212.6 1078.23   224.6 1077.98   244.7 1079.49   292.9 1080.23
   317.5 1081.93   337.1 1082.03   369.2 1082.95   389.3 1083.92   449.4 1085.73
   493.5 1087.91   505.5 1089.32   521.5 1093.03   525.5 1093.53   536.1 1093.97
#Mann= 6 ,-1,0
       0      .1       0  170.62     .05       0   189.6    .045       0
   209.7     .05       0   361.5     .06       0  461.23     .05       0
Bank Sta=189.6,209.7
XS Rating Curve= 0 ,0
Exp/Cntr=0.3,0.1

Type RM Length L Ch R = 1 ,13580   ,184.2,176.9,174.4
XS GIS Cut Line= 4
2175238.87126417753152.4158462392175203.93972654753278.834744324
 2175097.4817071 753370.322104782175045.08440065753468.463091451
#Sta/Elev= 30
       0 1099.46    46.4 1087.19      63 1082.33    71.3 1080.52    79.6 1079.37
    92.1  1078.5   108.7 1078.16   125.3 1077.36   146.7 1077.59   162.5  1077.2
   169.5 1076.48   172.4 1076.54     178 1077.47   188.9 1077.25   199.4 1077.76
   203.6 1077.53   212.1 1076.47   216.11076.159   223.4 1075.65   225.8 1075.69
   227.51076.186   231.9 1077.66   236.3 1078.07   277.6 1077.74   283.8  1078.1
   297.4 1079.38   306.5 1080.53   342.8 1086.45   362.8 1089.27   382.8 1091.65
#Mann= 5 ,-1,0
       0      .1       0      60     .05       0   216.1    .045       0
   227.5     .05       0  231.16     .06       0
Bank Sta=216.1,227.5
XS Rating Curve= 0 ,0
Exp/Cntr=0.3,0.1

Type RM Length L Ch R = 1 ,13403   ,156.7,150,153.4
XS GIS Cut Line= 4
2175085.00615794753124.969638102     2175039.174      753194.116
2175019.30159907753225.6057346042174892.88270099 753505.88973891
#Sta/Elev= 30
       0 1096.47      53 1085.37    57.8  1082.6    62.6 1077.15    65.61075.896
    67.4 1075.42    72.9 1075.35    81.8 1075.37   86.86 1075.89    91.3 1077.17
      96 1077.41   146.1 1076.33   167.6 1077.33   189.9 1077.34     225 1078.34
   277.7 1078.27   286.5 1079.43   295.2  1081.5     304 1084.66   312.8 1089.42
   317.2 1090.89   321.8 1091.79     326 1092.39   334.7 1092.68   352.3  1091.8
   361.1 1094.63   369.8 1095.64   378.6 1097.59   404.9 1099.35   427.7 1103.05
#Mann= 5 ,-1,0
       0     .05       0    65.6    .045       0   86.86     .05       0
  102.96     .06       0  320.19     .05       0
Bank Sta=65.6,86.86
XS Rating Curve= 0 ,0
Exp/Cntr=0.3,0.1

Type RM Length L Ch R = 1 ,13253   ,216.1,217,213.7
XS GIS Cut Line= 3
2174984.82299176752989.328987497     2174894.837      753170.338
2174753.60948079753434.290240625
#Sta/Elev= 30
       0 1117.17    17.7 1113.13    57.9  1102.6   124.9 1087.98   131.5 1085.86
   147.2 1079.02   151.7 1077.61   160.6 1076.88   178.5 1077.48   188.3 1075.98
   196.4  1075.7   209.9  1075.1  216.52 1075.71   223.5 1076.72   237.1 1075.83
   271.2  1077.9   314.2 1076.92   336.2 1077.02   348.1 1077.87   362.8  1081.2
   368.8 1083.86   377.6 1089.23   382.3 1090.66   395.9  1091.3   410.1 1090.62
     419 1094.23   427.9  1094.8   441.3 1098.94   470.6 1105.25   501.5 1111.19
#Mann= 5 ,-1,0
       0     .05       0     140     .06       0   196.4    .045       0
  216.52     .06       0  362.14     .05       0
Bank Sta=196.4,216.52
XS Rating Curve= 0 ,0
Exp/Cntr=0.3,0.1

Type RM Length L Ch R = 1 ,13036   ,223.8,222.9,214.5
XS GIS Cut Line= 2
2174829.65654757752843.8189984332174617.67683089 753267.15026195
#Sta/Elev= 30
       0 1109.98    61.7 1099.46    74.8 1097.72   127.3 1089.55     176 1082.58
   204.8 1079.59   220.7 1076.77  229.56 1075.72   238.6 1074.62   247.6 1075.72
   271.3 1076.47   287.8  1076.4   305.7 1076.84     346 1076.19   359.8 1076.57
   381.8 1076.27   390.7 1076.87   395.2 1077.63   399.7 1079.14   410.5 1086.04
   413.5 1087.65   416.5 1088.61     422 1089.33     431 1089.66   444.4 1089.08
   448.9 1090.84   455.2 1094.35   461.2 1096.88   467.1 1098.65   473.4 1099.67
#Mann= 5 ,-1,0
       0     .05       0  229.56    .045       0   247.6     .05       0
     300     .06       0     420     .05       0
Bank Sta=229.56,247.6
XS Rating Curve= 0 ,0
Exp/Cntr=0.3,0.1

Type RM Length L Ch R = 1 ,12813   ,134.9,138.9,142.6
XS GIS Cut Line= 4
2174704.41953706752705.6030550482174532.94491084752922.256624703
2174504.19467411753043.418336643 2174395.3544922753150.204930216
#Sta/Elev= 30
       0  1113.6     9.7 1112.43    28.3 1108.24    50.5 1105.78   106.6  1097.2
   152.5 1087.86   203.5 1080.82   219.5 1077.67   233.4 1076.63   258.2  1076.2
   339.2 1076.58   345.1 1075.64  349.49 1073.72   357.4 1072.22   361.5 1072.48
   365.11073.725     378 1075.23   424.7 1075.14   438.9 1076.05   445.7 1077.87
   454.7 1081.46   460.5 1084.25   467.1 1088.44   471.9 1090.17   483.3 1090.38
   500.4 1088.81   503.9 1090.33   512.9 1097.38   517.6 1099.99   553.3 1106.53
#Mann= 9 ,-1,0
       0     .05       0     100     .07       0     140     .05       0
     260     .07       0     270     .05       0  349.49    .045       0
   365.1     .05       0   376.3     .06       0  490.83     .05       0
Bank Sta=349.49,365.1
XS Rating Curve= 0 ,0
Exp/Cntr=0.3,0.1

Type RM Length L Ch R = 1 ,12674   ,66.9,68.4,69.8
XS GIS Cut Line= 3
2174673.50058989752648.3937667592174629.46311212752707.481098658
2174267.80338816 753110.21258938
#Sta/Elev= 30
       0 1117.56      11  1115.4    45.9 1106.13    65.8 1104.69    95.6 1099.99
   145.9 1094.64   189.1 1087.87   223.1 1083.85   257.1 1081.46   350.2 1078.85
     369 1076.06   390.2 1074.91   398.5 1073.86   404.9    1074   409.3 1073.24
   414.7 1072.27   428.8 1071.99   434.8 1072.27   437.9 1073.28   446.9 1077.36
   468.4 1081.12   486.5 1087.66     495 1089.66   522.2 1091.72     546 1090.33
   551.7 1092.54   560.5 1098.32   565.8 1101.03   602.7 1105.89     615 1108.25
#Mann= 7 ,-1,0
       0     .05       0   93.69     .07       0  203.69     .06       0
  223.69     .07       0   409.3    .045       0   437.9     .07       0
  483.69     .05       0
Bank Sta=409.3,437.9
XS Rating Curve= 0 ,0
Exp/Cntr=0.3,0.1

Type RM Length L Ch R = 1 ,12606   ,210,212.5,214.6
XS GIS Cut Line= 3
2174622.71250087752597.1821766762174252.65923054753037.129915792
2174206.42109751 753089.53585632
#Sta/Elev= 30
       0 1119.14   126.7 1094.58   177.7 1088.55   194.8 1082.89   203.4 1081.39
   219.5 1080.34   240.1 1080.07     277 1078.38   334.5 1077.69   396.4 1076.06
   401.6 1075.18  410.08 1072.77   419.1 1071.78   424.8 1071.86   430.5 1072.77
   441.8 1076.32   454.7 1079.56   465.2 1081.64   473.1  1082.3   488.6 1085.79
   494.9 1086.69   519.7 1089.49   549.7  1092.1   564.5 1091.74   580.3 1089.86
     591 1095.28   596.3 1099.02   601.6 1101.57   623.4 1105.45   644.8 1108.44
#Mann= 7 ,-1,0
       0     .05       0     130     .06       0     280     .05       0
     290     .06       0  410.08    .045       0   430.5     .06       0
     550     .05       0
Bank Sta=410.08,430.5
XS Rating Curve= 0 ,0
Exp/Cntr=0.3,0.1

Type RM Length L Ch R = 1 ,12394   ,332.2,320.1,304.2
XS GIS Cut Line= 5
2174418.82100682752567.9345909552174367.17612406752613.319487923
2174257.62637276752722.8692392242174184.07153975752787.034093557
2174119.90668541753040.563517997
#Sta/Elev= 30
       0 1100.75    20.1 1099.15    46.1 1095.53    93.4 1087.59   108.2 1083.04
   127.3 1082.75   166.9 1076.44   183.9 1075.82   245.4 1076.06   257.5 1074.98
   268.1 1072.67   275.9 1072.54   285.9 1071.81  295.36 1072.54   305.2 1075.52
   321.2 1077.87   339.4 1077.97   369.1 1076.98   421.8 1080.04   459.7 1083.83
   488.5 1087.66   505.1 1088.72   521.6 1091.98   533.9 1093.44   542.2 1093.39
   558.7 1091.64   562.8 1091.71   571.1  1094.7   579.3 1100.29   582.8 1101.58
#Mann= 7 ,-1,0
       0     .07       0   78.75     .05       0   275.9    .045       0
  295.36     .05       0  351.29     .06       0  461.29     .07       0
  561.29     .05       0
Bank Sta=275.9,295.36
XS Rating Curve= 0 ,0
Exp/Cntr=0.3,0.1

Type RM Length L Ch R = 1 ,12073   ,142.2,136.8,131.2
XS GIS Cut Line= 3
2173969.98496335752201.3508106882174078.43921714 752935.17764476
 2174055.9032683753049.265885758
#Sta/Elev= 30
       0 1093.39    15.9 1095.63    32.2  1096.9    76.7 1099.14   141.3 1099.21
     198 1096.63   242.4 1091.97     295 1090.59   304.7 1089.25   311.2 1086.89
   323.3 1075.61   327.3 1072.92   329.81072.024   335.4 1071.22   343.5 1071.31
   347.6    1072   359.7 1075.11     388 1076.51   432.5 1075.81   485.9 1076.25
   579.5 1075.64     667 1076.52   764.2 1086.79   792.8  1092.7   800.9 1093.81
   813.2 1093.34   825.4 1091.98   829.5 1092.22   849.8 1099.93   858.1 1100.66
#Mann= 5 ,-1,0
       0     .05       0   329.8    .045       0   347.6     .05       0
     720     .07       0   821.8     .05       0
Bank Sta=329.8,347.6
XS Rating Curve= 0 ,0
Exp/Cntr=0.3,0.1

Type RM Length L Ch R = 1 ,11937   ,187.1,190,197.3
XS GIS Cut Line= 3
2173679.37223992752215.1169338252173949.71523884752681.579650354
2173962.06086467753062.754416247
#Sta/Elev= 30
       0 1083.15    73.4 1081.13   182.7 1079.27   221.6 1078.01   248.9 1075.35
   261.3 1077.17   321.1 1077.78   347.5 1077.29   392.5 1075.07   404.6 1075.14
   409.2 1074.51   416.4 1072.28   427.7  1071.4  438.54 1072.28   450.8 1074.79
   515.6  1076.7   650.8 1074.81   674.8 1075.52   710.8 1074.64   750.9 1074.79
   762.9 1075.36   778.9 1076.95   814.9 1084.45   830.9 1086.88   850.5  1092.5
   858.9 1094.34   866.8 1094.38   886.9 1092.69   904.3 1095.79   920.5 1099.45
#Mann= 7 ,-1,0
       0     .05       0     130     .06       0     160     .05       0
   416.4    .045       0  438.54     .05       0  779.14     .06       0
  879.14     .05       0
#XS Ineff= 2 , 0
          342.54 1084.66
Permanent Ineff=
       T       F
Bank Sta=416.4,438.54
XS Rating Curve= 0 ,0
Exp/Cntr=0.3,0.1

Type RM Length L Ch R = 1 ,11747   ,88.6,91.1,93.3
XS GIS Cut Line= 4
2173584.57620758752331.3534973822173807.83521196752698.248763634
2173829.39788951752841.9999472912173859.82142044753091.815165663
#Sta/Elev= 30
       0 1082.39     167  1078.1   306.7 1076.97   359.1 1075.81   368.6 1075.38
   382.4 1071.95   385.3 1072.32   391.7 1074.65   414.7 1076.88     426 1075.37
   460.5 1072.33   468.9 1071.28   476.9 1071.53   480.2 1072.36     485 1074.37
   489.1 1075.04     570 1074.94   614.3 1074.27   658.6 1075.08   674.8 1077.25
   698.9 1082.78   731.1 1088.01   745.4 1092.54   755.3 1095.02   763.4 1095.59
   783.6 1093.72   787.6 1094.51   799.7 1099.63   811.8 1100.88   826.5 1103.34
#Mann= 7 ,-1,0
       0     .06       0     110     .05       0     150     .06       0
     230     .07       0  449.48     .06       0   460.5    .045       0
   480.2     .06       0
#XS Ineff= 2 , 0
        282.2155  1087.4
Permanent Ineff=
       T       F
Bank Sta=460.5,480.2
XS Rating Curve= 0 ,0
Exp/Cntr=0.3,0.1

Type RM Length L Ch R = 1 ,11656   ,50.7,52.9,53.2
XS GIS Cut Line= 6
2173540.91167207752374.697557437 2173686.1313982752595.084165958
2173721.09521857752670.9960870732173726.63990708752712.581250917
2173725.14957662752793.460799405 2173626.5773364753159.820958896
#Sta/Elev= 30
       0 1087.18    53.2 1083.45   105.2  1081.4   220.7 1078.73   307.1 1075.94
   327.4 1075.92   345.3 1074.75   402.1 1075.96   406.1 1075.59   422.1 1071.83
   426.1 1071.16   436.5 1070.97   443.9 1071.84   450.1 1073.78   458.1 1074.82
   515.4 1074.89   563.3 1074.12   597.9 1074.47   623.8 1075.86   650.1 1078.71
   685.1 1079.37   697.6 1080.66   709.7 1083.68   754.4 1091.66   768.4 1093.54
   784.8 1094.84   797.2 1098.22   805.5 1099.33     818 1100.34   849.8 1100.31
#Mann= 9 ,-1,0
       0     .05       0      40     .06       0      60     .05       0
     220     .07       0  293.93     .05       0   422.1    .045       0
   443.9     .05       0  500.37     .07       0  597.52     .06       0
#XS Ineff= 2 , 0
        264.5811  1087.4
Permanent Ineff=
       T       F
Bank Sta=422.1,443.9
XS Rating Curve= 0 ,0
Exp/Cntr=0.3,0.1

Type RM Length L Ch R = 1 ,11603   ,238.6,227.5,217.5
XS GIS Cut Line= 6
2173514.57268472752391.010867194 2173667.5650159 752626.14673189
2173672.69898674752663.1113219742173677.83295759752723.692177943
2173668.59181006752825.3448006722173585.42148238753152.892140576
#Sta/Elev= 30
       0 1087.54    54.3 1082.88      98 1081.06     156 1080.34   169.6  1081.3
   179.2 1080.09   212.6 1079.66     234 1081.76     267 1081.51   274.5  1080.7
   283.6 1078.14     314 1076.18   360.1 1075.54   392.2  1076.2   403.41071.798
   416.3 1070.89   424.81071.797   428.3 1073.51   432.4 1074.42   448.4 1075.33
   498.7 1074.51   596.2 1074.53   612.6 1075.81     658 1075.19   673.5    1076
   740.5 1085.15   761.2  1090.5     775 1096.19   785.9 1099.31   818.7 1102.63
#Mann= 8 ,-1,0
       0     .05       0     270     .07       0     280     .05       0
   403.4    .045       0   424.8     .05       0  478.64     .07       0
  530.72     .05       0  680.72     .06       0
Bank Sta=403.4,424.8
XS Rating Curve= 0 ,0
Exp/Cntr=0.3,0.1

Type RM Length L Ch R = 1 ,11375   ,172.4,177,178.5
XS GIS Cut Line= 4
2173331.04008353752405.6560401872173539.52493513752899.327267808
2173609.75765629752979.725251239 2173544.3850942753187.160491021
#Sta/Elev= 30
       0 1098.89    24.9 1097.16    29.9 1095.16    43.2 1088.06    61.6 1085.51
      82 1080.25    85.2 1079.98   101.2  1080.3     234 1078.97     260 1077.03
   305.8 1076.49   342.2 1076.75     412 1078.57   490.1 1078.94   519.5 1077.55
   543.3 1074.83     566 1074.27   585.9 1072.27   602.9 1070.44   608.5 1070.99
   612.7 1072.33     617 1073.69   623.3 1074.44   665.1 1074.33   702.9 1075.66
   752.7 1082.07   807.7 1094.02   832.9 1103.13   837.1 1104.12   860.1 1106.09
#Mann= 5 ,-1,0
       0     .05       0   585.9    .045       0   612.7     .05       0
  682.64     .06       0  812.64     .05       0
#XS Ineff= 2 , 0
        485.6098 1083.47
Permanent Ineff=
       T       F
Bank Sta=585.9,612.7
XS Rating Curve= 0 ,0
Exp/Cntr=0.3,0.1

Type RM Length L Ch R = 1 ,11198   ,212.6,221.3,225.4
XS GIS Cut Line= 3
2173148.32193975752587.0610524932173515.56640452753144.354582999
 2173536.1022879753261.865471227
#Sta/Elev= 30
       0 1082.48   136.7 1079.32   198.9 1079.18   241.1 1076.52   268.7 1073.83
   284.4 1073.18   498.1  1074.6   505.5 1074.11   512.5  1072.1   524.1 1071.17
   532.21072.028   561.6 1074.27   593.4 1073.48   606.1 1073.65   616.5  1074.6
   630.1 1078.49   646.7 1086.57   672.3 1097.42   676.4 1098.75   684.5 1099.96
   692.6 1103.71   699.8 1106.11     721 1107.74   730.9 1107.49   737.3 1106.27
   740.7 1106.57   749.5  1111.3   757.6 1114.14   765.7 1115.81   786.7 1118.55
#Mann= 4 ,-1,0
       0     .05       0   512.5    .045       0   532.2     .05       0
  737.42     .07       0
Bank Sta=512.5,532.2
XS Rating Curve= 0 ,0
Exp/Cntr=0.3,0.1

Type RM Length L Ch R = 1 ,10977   ,206.5,204.8,200.9
XS GIS Cut Line= 4
2173129.63288166752728.7287057562173243.00840989752905.644530148
 2173294.9819419753246.6416060192173308.92606025753359.462199894
#Sta/Elev= 30
       0 1082.94    57.5 1081.96   100.3 1078.43   128.8 1077.48   164.3 1073.03
     238 1073.89   270.4 1072.85   371.5 1072.52   420.1  1074.3   424.1 1073.28
   427.8 1070.92   436.2  1070.3     446 1070.98   452.4 1072.42   468.6 1073.33
   472.7 1074.49   492.9 1084.56   513.1 1097.01   537.4 1106.32   553.6 1107.94
   577.8 1113.17   589.9 1116.52   601.5 1122.04     605 1122.83     614  1123.5
   634.2 1122.49   637.3 1122.89   642.3 1125.36   654.3 1133.17   668.7 1139.26
#Mann= 4 ,-1,0
       0     .05       0   427.8    .045       0     446     .05       0
  625.06     .06       0
Bank Sta=427.8,446
XS Rating Curve= 0 ,0
Exp/Cntr=0.3,0.1

Type RM Length L Ch R = 1 ,10772   ,252.2,271.2,284.2
XS GIS Cut Line= 2
2172941.74276116752778.8530010772173175.16929168753423.472293467
#Sta/Elev= 30
       0 1082.02    74.8 1081.09   100.3 1078.86   130.1 1077.27   155.6 1073.66
   172.6 1072.46   253.6 1071.72   381.1 1073.99   387.9 1071.32   406.6 1070.25
   410.9 1071.27   415.1 1072.86   437.8 1073.79   444.9 1074.72   453.5 1077.54
   475.3 1086.77   483.2 1088.93   491.7 1090.01   517.2 1091.29   525.3  1092.6
   578.4 1109.15   589.6  1113.5   623.6 1118.62   629.8 1120.78   640.6 1126.26
     644 1127.22   653.4 1127.53   675.2 1125.96   678.9 1127.65   685.6 1132.79
#Mann= 4 ,-1,0
       0     .05       0   387.9    .045       0   410.9     .05       0
     670     .07       0
Bank Sta=387.9,410.9
XS Rating Curve= 0 ,0
Exp/Cntr=0.3,0.1

Type RM Length L Ch R = 1 ,10501   ,202.1,173.9,154.9
XS GIS Cut Line= 4
2172916.73290725752773.944662733 2172911.4239797753134.602290147
2172811.26256738753235.785757695 2173034.2018669753522.931296619
#Sta/Elev= 30
       0 1081.04    35.2 1081.94   139.2  1080.2   159.3 1078.79   183.3 1074.38
   203.3 1073.29   347.8 1073.58   410.8 1072.48   420.6 1071.33   429.9 1071.82
  435.26 1071.11   439.2 1070.38   444.9 1070.14   450.6 1070.31   454.4 1071.12
     462 1072.55   471.3 1072.95   570.7 1073.69   585.9 1074.56   602.4 1076.53
   621.3  1079.1   636.5 1081.86   697.3 1095.49   804.6 1115.14   818.8  1118.3
   839.1 1120.01     844  1121.3   850.3 1123.95   858.2 1124.59   866.6  1124.3
#Mann= 4 ,-1,0
       0     .05       0  435.26    .045       0   454.4     .05       0
  843.07     .07       0
Bank Sta=435.26,454.4
XS Rating Curve= 0 ,0
Exp/Cntr=0.3,0.1

Type RM Length L Ch R = 1 ,10327   ,38.4,36,36.4
XS GIS Cut Line= 6
 2172554.5084823 752791.196053082172613.10904084 752994.21710352
2172763.67650094753212.9894129962172714.46643442753337.907274165
2172833.07531271753437.589203785 2173016.3698631753544.025832732
#Sta/Elev= 30
       0  1088.2      27  1086.2    35.4  1086.4      52 1085.63    64.5 1084.29
   154.8 1077.61   185.2 1076.04   243.4 1074.08   309.4 1073.29   349.2 1073.53
   375.8 1072.13   388.9 1070.48   398.5 1069.62   413.8 1069.85  416.72 1070.46
   428.7 1072.17   473.5 1073.23   601.6 1073.18     643 1074.65   677.1 1077.43
   738.9 1084.22   793.5 1091.27   830.5 1096.96     906 1109.59   921.9 1110.78
   937.9 1113.23   950.7 1118.57   963.6 1122.64   973.9 1123.33   983.3 1123.23
#Mann= 6 ,-1,0
       0     .06       0      30     .05       0   388.9    .045       0
  416.72     .05       0  911.39     .06       0  931.39     .07       0
#XS Ineff= 2 , 0
        257.0772  1091.8
Permanent Ineff=
       T       F
Bank Sta=388.9,416.72
XS Rating Curve= 0 ,0
Exp/Cntr=0.3,0.1

Type RM Length L Ch R = 1 ,10291   ,189.7,188,183.1
XS GIS Cut Line= 6
2172496.12002573752804.543317442 2172559.0147238752995.219739698
 2172719.6122261753196.7509826072172670.30355421 753325.28930839
2172696.80128234753368.1903920242173004.79540492753595.529747169
#Sta/Elev= 30
       0 1092.03    35.4 1089.77    51.2 1087.75   110.2 1082.83   190.6 1078.65
   213.5  1074.6   254.4 1075.53   300.5 1073.26   407.9 1073.19   416.5 1072.45
  422.72 1070.29   430.7 1069.31   442.1  1069.4   447.8 1070.28   453.5 1072.37
   458.5 1072.69     574 1072.53   598.3 1072.92   665.8 1076.09   681.7 1075.78
   765.5  1084.5   823.2 1091.83   937.2 1109.06   975.4  1114.3   982.2 1115.86
   990.9 1119.78   994.5 1120.89  1004.1 1121.41  1022.7 1120.93  1033.5 1121.33
#Mann= 8 ,-1,0
       0     .06       0      20     .05       0     120     .06       0
  230.78     .05       0  422.72    .045       0   447.8     .05       0
  879.73     .06       0  999.73     .07       0
#XS Ineff= 2 , 0
        268.1557  1091.8
Permanent Ineff=
       T       F
Bank Sta=422.72,447.8
XS Rating Curve= 0 ,0
Exp/Cntr=0.3,0.1

Type RM Length L Ch R = 1 ,10103   ,133.1,136.3,135.4
XS GIS Cut Line= 3
     2172294.009      753059.199     2172639.056      753342.484
2172941.82717806753659.004881656
#Sta/Elev= 30
       0 1124.47    33.9 1118.08    44.2 1115.21    85.6 1109.88   121.8 1102.66
   183.9 1092.93   221.8 1085.91   274.2 1080.97   298.5 1073.85     307 1072.17
   328.9  1071.8   419.2 1072.92  431.77 1070.74   448.1 1069.86   453.8 1070.73
   459.6 1071.68   472.3 1071.41   483.4 1073.21   505.7 1074.56   549.8 1076.46
   647.2 1086.38   754.6 1098.92   794.3 1102.41     810 1104.62   833.9 1109.57
   839.6 1111.81     848 1116.76   850.9 1117.43   876.3 1118.34   884.5  1119.9
#Mann= 4 ,-1,0
       0     .05       0  431.77    .045       0   453.8     .05       0
  786.44     .06       0
Bank Sta=431.77,453.8
XS Rating Curve= 0 ,0
Exp/Cntr=0.3,0.1
